HEC-RAS study SWTSPRNGSCK.prj: SWTSPRNGSCK

--- SWTSPRNGSCK.g01 (geometry) --- (continued)

Type RM Length L Ch R = 1 ,23106   ,41.1,41.1,41.1
XS GIS Cut Line= 4
      2174746.92      220110.016     2174663.586      219776.682
     2174668.795      219719.391      2174746.92      219394.738
#Sta/Elev= 30
       0 2265.94    35.8 2260.51    76.4 2253.41    90.6 2250.27   140.7 2244.22
   166.4 2239.92   242.1  2238.4   275.9 2242.06   306.4 2243.16     337 2240.13
   343.6 2238.43   351.1  2234.2   356.42232.103   366.6 2230.76   373.2 2230.88
  377.862232.057   383.1 2233.94   396.1 2232.93   446.8 2233.12   544.6 2231.46
   571.6 2231.68   595.3 2233.11   615.5 2233.42   625.6 2234.42   642.5 2234.47
   649.2 2233.42     656 2234.75   666.1 2240.63   720.1 2250.21     735 2252.09
#Mann= 5 ,-1 , 0
       0    .035       0   356.4    .045       0  377.86    .035       0
  541.12     .06       0  641.12    .035       0
#XS Ineff= 2 ,-1
       0  351.34 2236.95  396.98   678.62238.717
Permanent Ineff=
       F       F
Bank Sta=356.4,377.86
XS Rating Curve= 0 ,0
Exp/Cntr=0.3,0.1

Type RM Length L Ch R = 1 ,23065   ,276.4,277.3,274.9
XS GIS Cut Line= 4
     2174795.531      220127.377     2174705.253      219771.474
     2174710.461      219714.182     2174781.642      219403.418
#Sta/Elev= 30
       0 2277.92    30.1 2273.97   112.3  2258.5   152.8 2251.45   199.3 2245.01
   233.8 2238.79   300.8 2236.28   314.4 2236.74   351.6 2235.55   365.2 2234.24
   372.42230.715   376.8  2229.6     385 2229.33   388.3 2229.85   389.62230.681
   394.9 2233.76   431.2 2231.77   488.5  2232.2   565.9 2230.52   589.5 2231.16
   616.4  2233.1   623.1 2232.81   636.6 2233.86   653.4 2233.96   663.4 2233.35
   666.8 2234.23   674.3 2238.54   679.8 2240.48   726.3 2249.78   743.5 2252.29
#Mann= 5 ,-1 , 0
       0    .035       0   372.4    .045       0   389.6    .035       0
   554.7     .06       0   654.7    .035       0
#XS Ineff= 2 ,-1
       0  363.312235.715  412.07  694.892237.385
Permanent Ineff=
       F       F
Bank Sta=372.4,389.6
XS Rating Curve= 0 ,0
Exp/Cntr=0.3,0.1

Type RM Length L Ch R = 1 ,22787   ,229.7,233.2,234.3
XS GIS Cut Line= 2
     2174953.517      220144.738     2174991.711       219420.78
#Sta/Elev= 30
       0 2281.84    36.7 2281.67    97.3 2282.91   112.3 2282.12   147.6 2278.82
   181.3 2273.94   220.7 2266.62     247 2260.52   283.1 2250.78   296.3 2246.06
   306.1 2241.67   322.8 2230.73     3282226.015   329.1 2224.93   332.4 2224.62
     339 2224.99   344.42226.395   352.1 2227.34     362 2227.51   387.9 2226.71
   424.4 2227.08   486.8 2225.76     572 2227.27   588.7 2229.58   595.2 2229.91
   614.9 2229.83   628.1 2228.71     650 2231.85   677.4 2233.91     725 2239.58
#Mann= 5 ,-1 , 0
       0    .035       0     328    .045       0   344.4    .035       0
     560     .06       0     660    .035       0
Bank Sta=328,344.4
XS Rating Curve= 0 ,0
Exp/Cntr=0.3,0.1

Type RM Length L Ch R = 1 ,22554   ,277.5,277.2,273.3
XS GIS Cut Line= 2
     2175108.101       220171.22     2175273.049      219447.985
#Sta/Elev= 30
       0 2258.34    24.4 2256.64    44.6 2256.41    95.1 2259.68   175.8 2268.08
   199.4 2269.15   219.6  2268.7   239.8  2265.7   256.6 2262.07   286.9 2254.53
   307.6 2248.49   317.1 2245.17   340.7 2234.41   367.6  2224.8  370.492223.106
   374.4 2221.55   384.5 2221.94   388.92223.284   404.6 2222.76   465.2 2223.53
   537.8 2222.75   556.1 2223.02   579.6 2225.49   593.1 2225.86   606.5 2225.64
   616.6 2224.49   623.4 2225.25   633.5 2224.44   663.8 2224.27   741.8 2227.83
#Mann= 6 ,-1 , 0
       0    .035       0  370.49    .045       0   388.9    .035       0
     500     .06       0     600    .035       0     700     .06       0
#XS Ineff= 2 , 0
                          592.18         2245.77
Permanent Ineff=
       F       F
Bank Sta=370.49,388.9
XS Rating Curve= 0 ,0
Exp/Cntr=0.3,0.1

Type RM Length L Ch R = 1 ,22277   ,234.7,244.7,254.7
XS GIS Cut Line= 3
     2175309.601      220236.947      2175434.42      219882.585
     2175469.142      219512.793
#Sta/Elev= 30
       0 2283.58    33.1 2279.64    60.1 2275.45      81  2271.1   174.6 2254.67
   223.4 2245.21   241.5 2242.39   251.4 2239.81   261.9 2238.18   272.2 2235.65
   293.2 2231.86     321 2228.14   341.5 2226.02   373.2 2223.52   393.1    2220
   401.82217.612   412.8 2217.23   427.8 2217.78   442.5  2219.3   551.2 2219.71
   567.7 2218.96   574.3 2219.21   587.5 2218.74     592 2219.19   603.8  2221.5
     627 2223.06   656.7 2222.26   673.2 2223.07   706.1 2223.54   747.1 2229.49
#Mann= 5 ,-1 , 0
       0    .035       0   401.8    .045       0   427.8    .035       0
   575.7     .04       0   675.7     .06       0
Bank Sta=401.8,427.8
XS Rating Curve= 0 ,0
Exp/Cntr=0.3,0.1

Type RM Length L Ch R = 1 ,22032   ,251,253,242.7
XS GIS Cut Line= 3
      2175361.53       220263.59     2175587.744      219974.227
     2175873.667      219689.943
#Sta/Elev= 30
       0 2292.82    49.5 2288.91   109.9 2276.72   143.3 2271.12   164.1 2266.77
   194.4 2259.54   251.5 2240.66   276.2 2233.76   306.5 2223.81   326.5 2219.99
     351 2217.63   360.72214.993   366.3 2214.38   377.12214.717   389.5  2215.3
   418.4 2214.79   432.3 2215.82   443.9 2215.88   495.9  2215.4   513.5  2214.5
   593.1 2212.95   614.9 2213.54   619.5 2214.48   624.8 2216.47   634.1 2217.65
   657.3 2218.49   671.8 2217.37   713.4  2223.4   736.5 2228.04   770.5 2232.93
#Mann= 5 ,-1 , 0
       0    .035       0   360.7    .045       0   377.1    .035       0
  627.29     .04       0  767.29     .05       0
Bank Sta=360.7,377.1
XS Rating Curve= 0 ,0
Exp/Cntr=0.3,0.1

Type RM Length L Ch R = 1 ,21779   ,279,284.4,284.9
XS GIS Cut Line= 3
     2175573.309      220332.238     2175739.975      220136.057
      2175924.35      219720.359
#Sta/Elev= 30
       0 2298.47      85 2274.58   117.6  2263.9   137.9 2258.49   160.7 2250.79
   173.5  2247.3   177.9  2245.7   203.7 2232.53   239.2 2220.06   257.3 2216.48
   282.1 2213.43   298.8 2211.92   322.82211.417   338.3 2208.73   341.9  2209.3
   345.82211.582     399 2212.78   435.2 2212.19   449.5 2211.19   485.4 2210.71
   524.9 2211.83   535.8 2213.04   558.1 2214.03   576.3 2216.37   592.9 2217.23
   602.9 2217.02     611 2219.62   618.2 2221.21   640.2 2222.98   712.2 2234.02
#Mann= 6 ,-1 , 0
       0    .035       0   322.8    .045       0   345.8    .035       0
  537.42     .04       0  587.42     .06       0  647.42     .05       0
Bank Sta=322.8,345.8
XS Rating Curve= 0 ,0
Exp/Cntr=0.3,0.1

Type RM Length L Ch R = 1 ,21495   ,211.8,212.6,211.7
XS GIS Cut Line= 2
     2175799.361      220460.843     2176241.271      219865.231
#Sta/Elev= 30
       0 2274.74    51.2 2253.43   100.8 2235.93   111.8 2231.07   156.7 2218.72
   177.8 2213.98   210.9 2209.83   239.1 2207.16   279.9 2206.31     329 2207.23
  361.37 2206.76   369.8 2204.79   376.1 2204.27   381.6 2205.33  383.572206.622
   388.9 2210.09   393.6 2211.49   418.8 2212.68   435.2 2214.74   492.4 2215.63
   529.6 2212.96   562.5 2213.12   569.5 2216.52   581.2 2225.58   586.3 2227.99
   602.7 2230.96   628.1 2233.24   689.1 2242.18   721.1 2246.19   741.6 2247.87
#Mann= 7 ,-1 , 0
       0    .035       0     350     .06       0  361.37    .045       0
  383.57     .06       0     450    .035       0     480     .06       0
     620    .035       0
Bank Sta=361.37,383.57
XS Rating Curve= 0 ,0
Exp/Cntr=0.3,0.1

Type RM Length L Ch R = 1 ,21282   ,249.5,250,245.7
XS GIS Cut Line= 3
     2175979.841      220566.361     2176193.848      220269.959
     2176407.231      219967.465
#Sta/Elev= 30
       0 2261.95    71.6 2236.07    98.7 2224.89   108.1  2222.7   140.4 2213.33
   164.6 2207.99   205.1 2204.89   245.6 2203.44   269.9 2203.91   300.7 2202.62
   349.1 2203.24   355.82202.903   368.9 2200.54   371.7 2200.73  377.722202.987
     383 2203.61   395.1 2203.39   483.4  2204.7   491.4 2206.08   500.7 2209.04
   511.5 2210.35   526.6 2210.76   543.1 2210.23   559.7 2212.33   567.7 2214.58
   575.7 2219.37   595.8 2223.47   622.1 2229.84   689.1 2248.08   735.8 2259.01
#Mann= 6 ,-1 , 0
       0    .035       0   355.8    .045       0  377.72    .035       0
  475.59     .04       0  495.59     .06       0  595.59    .035       0
#XS Ineff= 2 , 0
                          438.84          2218.3
Permanent Ineff=
       F       F
Bank Sta=355.8,377.72
XS Rating Curve= 0 ,0
Exp/Cntr=0.3,0.1

Type RM Length L Ch R = 1 ,21032   ,245.2,249.4,254.7
XS GIS Cut Line= 3
      2176226.27      220697.723     2176404.505       220381.55
     2176586.754      220057.555
#Sta/Elev= 30
       0 2250.04    54.7 2230.33    74.4  2222.5    88.9 2217.94    98.5 2213.94
   134.8 2205.91   149.6 2203.44   187.3 2200.73   258.8 2199.75   288.8 2198.55
   353.1 2199.37   360.5 2196.95   364.3 2197.14     3762199.487   398.2 2199.45
   416.5 2200.34   447.8 2199.96   454.6 2202.06   462.2 2206.36   477.2 2208.05
   500.8 2207.89   518.6 2204.88   526.2 2204.37   541.2 2204.28   562.8 2206.04
   580.3 2208.53   623.7 2216.55   650.2 2223.16   699.3 2238.27   734.7 2247.03
#Mann= 5 ,-1 , 0
       0    .035       0   353.1    .045       0     376    .035       0
  482.95     .06       0  592.95      .1       0
#XS Ineff= 2 , 0
                           417.8         2205.57
Permanent Ineff=
       F       F
Bank Sta=353.1,376
XS Rating Curve= 0 ,0
Exp/Cntr=0.3,0.1

Type RM Length L Ch R = 1 ,20783   ,256.3,257.8,253.5
XS GIS Cut Line= 3
     2176404.906       220827.03      2176536.85      220583.974
     2176870.184      220261.057
#Sta/Elev= 30
       0 2261.81    19.2 2259.71    34.1 2257.29    71.4 2249.17   108.8 2237.76
   135.2 2228.35   146.1 2223.73   168.5 2217.07   179.7 2213.17   198.4 2207.97
   220.8 2202.84   239.4 2199.98   258.1 2198.35   347.4 2194.43   358.52194.356
   370.3 2192.97   384.42194.953   397.7 2194.96     423    2196   456.5 2203.07
   475.3  2205.1   502.8 2204.81   521.5 2202.81   542.4 2202.26   572.6  2202.9
   607.4 2207.65   639.8 2214.31   680.9 2220.68   702.5 2222.89   740.7  2227.8
#Mann= 6 ,-1 , 0
       0    .035       0   358.5    .045       0   384.4    .035       0
  436.56     .04       0  586.56      .1       0  716.56     .06       0
Bank Sta=358.5,384.4
XS Rating Curve= 0 ,0
Exp/Cntr=0.3,0.1

Type RM Length L Ch R = 1 ,20525   ,185.2,187.1,185.3
XS GIS Cut Line= 3
     2176429.211      220854.807     2176741.711      220731.543
     2177014.281      220443.349
#Sta/Elev= 30
       0 2254.22    32.9 2249.74    98.5 2242.38   130.6 2237.14     181 2227.62
   257.8 2217.16   293.9 2213.72   325.6 2208.61   341.1 2206.84   345.5 2205.87
   350.6 2203.18   364.9 2197.89   375.32191.768   379.3 2190.55   387.2 2189.58
   393.6 2189.85   401.52191.325   456.9 2192.43   498.6 2191.38   503.2 2192.08
   516.7 2199.77   525.7 2201.48   547.4 2201.78   563.6  2200.3   577.6 2201.45
   622.8 2209.83   635.6 2213.36   658.8 2218.36   703.9 2230.89   732.6 2236.87
#Mann= 5 ,-1 , 0
       0    .035       0   375.3    .045       0   401.5    .035       0
  505.93     .04       0  645.93      .1       0
Bank Sta=375.3,401.5
XS Rating Curve= 0 ,0
Exp/Cntr=0.3,0.1

Type RM Length L Ch R = 1 ,20338   ,309.1,305.6,299.4
XS GIS Cut Line= 5
 2176783.9063114221162.5189090592176826.00258417220901.638000542
2176898.62237493220833.236485506 2176958.6050312220767.153898085
     2177173.537      220594.687
#Sta/Elev= 30
       0 2246.99    41.2 2239.81      91 2232.51   107.6 2229.33   157.5  2221.5
   190.7 2215.42     214 2210.37   260.5  2201.9   306.6 2196.21   315.6 2194.32
   332.2 2189.08   338.1 2188.12  343.78 2188.02   354.6 2186.93  365.242188.364
   381.9 2189.21   434.3 2189.48   462.3 2190.18   480.9 2191.55   511.3 2194.65
   546.3 2199.46   573.2 2199.71     579 2201.31   583.5 2203.42   591.9 2208.69
   596.1 2210.37   609.9 2211.96   625.6 2215.87     677 2227.22   728.8  2237.7
#Mann= 7 ,-1 , 0
       0      .1       0     100    .035       0  343.78    .045       0
  365.24    .035       0  453.26      .1       0  573.26     .04       0
  603.26      .1       0
#XS Ineff= 2 , 0
                          494.33         2210.98
Permanent Ineff=
       F       F
Bank Sta=343.78,365.24
XS Rating Curve= 0 ,0
Exp/Cntr=0.3,0.1

Type RM Length L Ch R = 1 ,20032   ,253.8,250,243.8
XS GIS Cut Line= 3
     2176959.772       221348.89     2177128.911      221027.402
     2177310.485      220707.201
#Sta/Elev= 30
       0 2296.81    19.3 2293.45    48.9 2286.75   108.3 2271.01   137.9 2260.59
   215.8 2236.68   264.3 2219.65   323.3 2200.62   338.1  2194.4   353.42185.261
   361.5 2183.18   376.32184.778   390.3    2186   458.4 2185.18   469.7  2186.4
   491.5 2193.44   522.8 2207.64   537.2 2212.67     542  2211.3   548.9 2204.48
   552.6 2199.73   556.4 2196.93   586.6 2197.18   590.4 2198.89   597.9    2206
   616.8 2220.66   631.9 2234.82   635.6 2236.86   646.9 2240.02   731.4 2257.16
#Mann= 5 ,-1 , 0
       0      .1       0   353.4    .045       0   376.3      .1       0
  433.27     .04       0  613.27      .1       0
Bank Sta=353.4,376.3
XS Rating Curve= 0 ,0
Exp/Cntr=0.3,0.1

Type RM Length L Ch R = 1 ,19782   ,243,250.7,259.6
XS GIS Cut Line= 3
     2177205.253      221438.141     2177356.295      221132.585
     2177427.475      220766.266
#Sta/Elev= 30
       0 2299.73    79.9 2275.35   136.9 2260.17   151.5 2255.06   171.9 2249.01
   190.9 2244.06   221.1 2237.57   235.7 2233.76   279.7 2216.75   301.7  2207.4
   319.9 2198.44   355.1 2183.23   361.8 2181.76   376.32181.292   385.2  2179.5
   388.5 2179.58   396.52181.568   447.3 2183.29   462.1 2184.91     478 2190.61
   492.3 2193.77   508.8 2194.91   532.3 2194.19   535.6 2194.82   545.6 2202.16
   555.7 2208.29     569 2218.92   599.1 2227.92   629.2 2235.11     714 2258.06
#Mann= 5 ,-1 , 0
       0      .1       0   376.3    .045       0   396.5      .1       0
  410.85     .04       0  610.85      .1       0
Bank Sta=376.3,396.5
XS Rating Curve= 0 ,0
Exp/Cntr=0.3,0.1

Type RM Length L Ch R = 1 ,19532   ,242.2,245.8,248.4
XS GIS Cut Line= 3
     2177323.765      221491.172     2177608.031      221177.724
     2177753.864      220917.307
#Sta/Elev= 30
       0 2293.39   105.8  2260.6   154.7 2247.76   204.9 2230.65   258.4 2214.63
   281.6  2205.7   315.8 2189.48   334.7  2181.5   367.42177.517   379.1 2175.75
   390.4    2178   398.8 2179.58   411.7 2179.99   414.4 2180.87   423.2 2186.48
   430.5 2188.81   454.6 2190.71   476.3 2190.76   487.2 2189.12     498 2184.97
   507.6 2184.64   512.5 2185.19   537.5    2193   573.7 2206.33     592 2214.41
     600 2217.07   607.5 2221.21     618 2225.14     694 2239.29   721.6  2245.2
#Mann= 6 ,-1 , 0
       0      .1       0     310     .12       0     330     .04       0
   367.4    .045       0   390.4     .04       0  493.15      .1       0
Bank Sta=367.4,390.4
XS Rating Curve= 0 ,0
Exp/Cntr=0.3,0.1

Type RM Length L Ch R = 1 ,19286   ,286.4,281.6,274.4
XS GIS Cut Line= 2
     2177441.147      221604.783     2178040.322       221170.78
#Sta/Elev= 30
       0 2286.24    80.1 2261.61    91.8  2256.6     120 2247.61   163.3 2235.73
   177.8  2230.8   191.3 2222.95   228.1 2210.16   250.7 2200.73   272.7 2190.79
   283.1 2183.31   286.8 2181.77   303.4 2178.03   360.1 2174.85   376.1 2173.38
     3832175.207   400.6 2176.81   425.4 2188.01   442.9 2192.08   465.4 2193.41
   469.5 2192.74   477.1  2187.8   481.6 2186.91   522.1 2186.83   526.8 2188.37
   538.2 2196.16   547.6 2203.89   552.3  2205.8   647.7 2217.11   739.8 2225.57
#Mann= 7 ,-1 , 0
       0     .12       0      10      .1       0     130     .12       0
   360.1    .045       0     383      .1       0     420     .04       0
     590      .1       0
Bank Sta=360.1,383
XS Rating Curve= 0 ,0
Exp/Cntr=0.3,0.1

Type RM Length L Ch R = 1 ,19004   ,164,161.6,158.9
XS GIS Cut Line= 3
     2177576.781      221792.307     2177901.434      221625.641
     2178112.572      221272.563
#Sta/Elev= 30
       0 2276.45    38.9 2265.21   105.3 2250.06   134.8 2240.41   160.6 2233.58
   197.5 2226.05   239.6  2214.5   312.2 2197.48   326.6 2192.93     345 2183.43
   367.7 2174.21   391.6  2171.6     4042171.286   412.9  2169.6   423.72170.908
   493.2 2172.17   508.5 2175.55     528 2182.49   550.5 2191.95   554.3 2191.13
   561.4 2185.02   565.8 2183.83   605.2 2184.19   607.9 2184.93   611.7 2187.83
   619.4 2197.68   630.8 2207.41   635.6 2210.39   714.9  2220.5   776.3 2225.86
#Mann= 9 ,-1 , 0
       0     .12       0      80    .035       0     190      .1       0
     404    .045       0   423.7      .1       0  434.93    .035       0
  444.93      .1       0  564.93     .04       0  674.93      .1       0
Bank Sta=404,423.7
XS Rating Curve= 0 ,0
Exp/Cntr=0.3,0.1

Type RM Length L Ch R = 1 ,18843   ,33.5,33.5,33.6
XS GIS Cut Line= 3
     2177712.197      221884.321      2178028.17      221755.849
     2178191.364       221335.71
#Sta/Elev= 30
       0 2227.63    44.5 2217.68    82.4 2210.03   252.4    2182   287.8 2177.58
   316.2 2176.76   358.9 2173.89   412.3  2171.8   415.9 2170.93   419.52168.857
   422.9 2167.34   427.8 2166.67   439.12168.807   458.2 2170.93   476.7  2170.5
   506.4 2172.19   517.9 2172.23     552 2178.53   595.4 2181.59     620  2181.7
   623.5 2183.46   633.1 2191.24   645.8 2200.38   655.2 2208.25   658.7 2210.06
   683.4 2214.98   697.4 2216.22     708 2218.45   781.9 2227.08   791.8 2227.32
#Mann= 8 ,-1 , 0
       0      .1       0      30    .035       0  361.09     .06       0
   419.5    .045       0   439.1     .06       0  451.09    .035       0
  561.09     .04       0  661.09      .1       0
#XS Ineff= 3 ,-1
       0  419.36 2170.85  452.04     4902170.849  490.24  539.97 2175.95
Permanent Ineff=
       F       F       F
Bank Sta=419.5,439.1
XS Rating Curve= 0 ,0
Exp/Cntr=0.3,0.1

Type RM Length L Ch R = 1 ,18809   ,206.6,206.9,209.2
XS GIS Cut Line= 3
     2177741.711      221915.571     2178055.947      221776.682
     2178220.878      221351.335
#Sta/Elev= 30
       0 2216.26    79.9    2202   159.7 2190.29   180.3    2186   234.1 2179.07
   302.3 2176.62   349.2 2176.64   412.5 2172.13   428.3 2169.59   437.1 2166.02
   444.2 2165.71  452.942169.585   500.5 2169.56   518.1 2170.67   532.1 2169.62
   535.7  2170.1   553.3 2176.91   556.8 2177.49     599 2180.77   622.7 2180.64
   627.2 2182.83   635.4 2190.29   658.2 2207.31   662.3 2209.07     687 2213.95
   724.1 2218.34   736.8 2218.97     747 2221.62   774.9 2224.88   799.8 2226.88
#Mann= 7 ,-1 , 0
       0    .035       0  373.56     .06       0   428.3    .045       0
  452.94     .06       0  473.56    .035       0  563.56     .04       0
  683.56      .1       0
#XS Ineff= 3 ,-1
  419.23  426.49 2170.42  454.36  509.09 2170.33  511.12  566.01 2175.26
Permanent Ineff=
       F       F       F
Bank Sta=428.3,452.94
XS Rating Curve= 0 ,0
Exp/Cntr=0.3,0.1

Type RM Length L Ch R = 1 ,18602   ,43.1,44,43.4
XS GIS Cut Line= 2
     2178111.503      222104.807     2178430.947      221438.141
#Sta/Elev= 30
       0 2233.25    34.9 2229.24   122.3 2213.92   155.4 2206.35     235 2182.79
   256.9 2178.45   283.3 2175.84   318.7 2175.74   351.5 2174.39   409.82166.541
   416.9 2162.77   420.6 2162.61     4352166.439     457 2166.55   464.2 2168.64
   477.6 2174.59   493.3 2175.79     512 2174.87   515.2 2174.03   526.1 2168.15
   534.1 2166.51     577 2167.16   593.2 2171.35   620.7 2180.69     635 2183.11
   660.7 2190.07   700.7 2198.77   711.6 2199.68   718.9 2202.36   739.2 2207.33
#Mann= 6 ,-1 , 0
       0    .035       0     390     .06       0   409.8    .045       0
     435     .06       0     500     .04       0     510      .1       0
#XS Ineff= 2 , 0
           409.8  2175.1     435          2175.1
Permanent Ineff=
       F       F
Bank Sta=409.8,435
XS Rating Curve= 0 ,0
Exp/Cntr=0.3,0.1

Type RM Length L Ch R = 1 ,18558   ,167.8,170.3,172.4
XS GIS Cut Line= 2
     2178149.697      222123.905     2178469.142      221457.238
#Sta/Elev= 30
       0    2239    34.3  2234.4    92.5  2224.1   110.7 2219.69   121.6 2218.71
   267.1 2175.99   345.2 2175.24     369 2173.25   394.5 2169.83   415.42165.273
   426.4 2162.38   430.8  2162.2   438.1 2162.95  443.282165.396   445.4 2166.23
   456.3 2167.68   470.6 2173.46   487.8 2174.56     500 2174.17   505.1 2173.29
   519.8 2166.62   525.4 2165.12   572.7 2165.18   587.3    2166   605.5 2170.36
     633 2182.64   638.2 2184.36   696.9 2195.92   707.3 2196.86   739.2 2205.28
#Mann= 5 ,-1 , 0
       0    .035       0     410     .06       0   415.4    .045       0
  443.28     .06       0     520      .1       0
#XS Ineff= 2 , 0
           415.4  2175.1  443.28          2175.1
Permanent Ineff=
       F       F
Bank Sta=415.4,443.28
XS Rating Curve= 0 ,0
Exp/Cntr=0.3,0.1

Type RM Length L Ch R = 1 ,18388   ,189.6,189.9,190.2
XS GIS Cut Line= 3
     2178243.442      222158.697     2178454.132      221861.412
     2178652.181      221556.086
#Sta/Elev= 30
       0 2250.18      48 2244.36    80.6 2239.26   113.9 2232.75     161 2221.06
   189.2 2215.85   213.3    2210   236.2 2207.11   293.7 2192.98     346 2176.24
     362  2169.5   377.5 2165.54   391.8  2163.5  394.872162.086   401.3 2158.78
   405.1  2158.6   413.1 2159.05   420.1 2162.21   428.6 2167.46   440.3 2169.57
   458.2 2169.73   473.7  2168.6   487.2 2164.08   503.3 2163.86   612.4 2169.73
   647.6 2176.78   702.3 2198.54   710.1 2204.26   714.1 2206.11   728.3  2209.4
#Mann= 5 ,-1 , 0
       0    .035       0  374.37     .04       0  394.87    .045       0
   420.1     .04       0  494.37      .1       0
#XS Ineff= 2 , 0
                          447.92         2169.69
Permanent Ineff=
       F       F
Bank Sta=394.87,420.1
XS Rating Curve= 0 ,0
Exp/Cntr=0.3,0.1

Type RM Length L Ch R = 1 ,18198   ,160.8,161.7,162.7
XS GIS Cut Line= 2
     2178415.322      222257.585     2178812.892      221665.571
#Sta/Elev= 30
       0 2242.21    99.8 2221.82   158.7 2207.23   246.9 2186.67   276.3 2181.75
   357.3 2170.17     362 2168.18   376.2 2157.41     381 2154.61     384 2154.04
     394 2154.73   399.12157.345   403.8 2161.91   405.8  2163.1   416.4 2164.84
   440.1  2164.7   455.2 2162.92     467 2160.54   482.6 2159.91   515.7 2161.24
   534.2 2163.22   570.6 2163.91   605.9  2167.5   617.2 2169.06   640.9 2174.38
   652.8 2176.05   660.7 2178.32   668.6 2179.52   680.4 2183.67   713.1 2191.94
#Mann= 5 ,-1 , 0
       0    .035       0     370     .04       0   376.2    .045       0
   399.1     .04       0     490     .06       0
#XS Ineff= 2 , 0
                          429.76         2164.95
Permanent Ineff=
       F       F
Bank Sta=376.2,399.1
XS Rating Curve= 0 ,0
Exp/Cntr=0.3,0.1

Type RM Length L Ch R = 1 ,18036   ,30.8,30.6,30.5
XS GIS Cut Line= 2
     2178524.697      222344.391      2178974.35      221750.641
#Sta/Elev= 30
       0 2210.92    39.6 2206.15    72.6 2201.03   159.8 2182.99   182.7 2177.17
     216 2170.79   262.9 2163.79     291 2160.74   328.5 2160.01   344.2 2157.54
   368.9 2157.91     373 2156.84   378.9 2153.98   385.3 2151.38   389.5 2150.63
   394.7 2151.51   398.82153.997   408.1 2158.89   416.4 2160.02   478.3 2160.01
   504.1 2161.59   514.2 2163.27   529.9 2167.99   546.8 2174.19   552.2 2175.22
   633.8 2179.95   689.9 2184.89   720.7 2186.62   731.6 2186.29   744.8 2187.91
#Mann= 6 ,-1 , 0
       0    .035       0     370     .06       0   378.9    .045       0
   398.8     .06       0     500      .1       0     620     .04       0
#XS Ineff= 2 , 0
           378.9  2159.3   398.8          2159.3
Permanent Ineff=
       F       F
Bank Sta=378.9,398.8
XS Rating Curve= 0 ,0
Exp/Cntr=0.3,0.1

Type RM Length L Ch R = 1 ,18006   ,221.2,223.3,224.1
XS GIS Cut Line= 2
     2178552.475       222358.28     2179002.128       221764.53
#Sta/Elev= 30
       0 2201.18    44.3 2196.59    84.4 2190.28   114.7 2184.07   139.4 2180.92
   180.2 2172.98   201.9 2170.07   234.5 2164.18   328.7 2157.21     356 2156.88
   365.4 2154.76   369.12153.089   375.8 2151.01   382.2 2150.23   386.3 2150.25
   393.82153.067   402.8 2158.47   406.9 2159.13   427.5 2159.88   446.5 2158.84
   460.4 2161.04   479.1 2159.44   484.5 2159.79   512.9 2172.33   552.7 2178.36
   593.2 2182.47   645.6 2184.78   707.3 2189.23   723.7 2193.64   744.8 2195.82
#Mann= 5 ,-1 , 0
       0    .035       0   369.1    .045       0   393.8     .06       0
     510      .1       0     640     .04       0
#XS Ineff= 2 , 0
          365.52 2158.14  394.82         2158.29
Permanent Ineff=
       F       F
Bank Sta=369.1,393.8
XS Rating Curve= 0 ,0
Exp/Cntr=0.3,0.1

Type RM Length L Ch R = 1 ,17782   ,259.7,256.5,247.3
XS GIS Cut Line= 3
     2178698.243      222472.712     2178944.507      222203.309
     2179190.235      221929.485
#Sta/Elev= 30
       0 2175.56    27.8 2173.98      70 2169.21   100.8 2167.77   112.6 2166.45
   141.1 2165.45   167.8 2161.81     190 2157.06   212.4 2155.26   234.4 2154.56
   252.2 2151.66   274.4  2153.2   327.8 2149.84   345.42147.157   367.8 2145.94
     3782147.607   387.9 2150.49   416.8 2153.41   433.1 2153.87   451.8 2153.28
   463.3 2156.63   482.4 2159.91   500.9 2162.19   565.5 2165.53     575 2166.54
   583.8 2168.53   610.2 2171.34     663 2181.14   697.4 2191.16   732.9 2205.31
#Mann= 9 ,-1 , 0
       0    .035       0     180      .1       0     340     .04       0
   345.4    .045       0     378     .04       0     445     .06       0
     485      .1       0     575     .06       0     625      .1       0
Bank Sta=345.4,378
XS Rating Curve= 0 ,0
Exp/Cntr=0.3,0.1

Type RM Length L Ch R = 1 ,17526   ,238.8,243.5,245.3
XS GIS Cut Line= 3
     2178932.788      222650.808     2179135.809      222363.488
      2179292.11      222010.579
#Sta/Elev= 30
       0 2213.48    32.2 2212.28     115 2204.76   156.8 2200.02   172.8 2199.12
   251.5 2184.51   261.2  2182.5   278.4 2177.46   305.4 2168.58   341.9 2153.02
   364.92144.322   371.2    2142   376.2 2141.45   378.7 2141.47   391.1 2144.43
   403.6  2144.6   421.6 2147.54   432.4 2148.08   446.7 2148.15   474.8 2146.83
   514.9 2146.93   579.5 2150.02     600  2152.8   622.4 2159.91   632.3 2167.08
   647.7 2171.37   662.5 2179.17     695 2189.29   715.8 2198.56   737.8 2207.25
#Mann= 5 ,-1 , 0
       0    .035       0     140      .1       0   364.9    .045       0
   391.1     .04       0  481.81      .1       0
#XS Ineff= 2 , 0
                          436.82         2166.63
Permanent Ineff=
       F       F
Bank Sta=364.9,391.1
XS Rating Curve= 0 ,0
Exp/Cntr=0.3,0.1

Type RM Length L Ch R = 1 ,17282   ,241,241.9,237.3
XS GIS Cut Line= 3
     2179113.386      222781.585     2179331.196      222457.816
     2179520.881      222152.778
#Sta/Elev= 30
       0 2229.69   149.8 2201.17   189.4 2196.64   213.1 2192.25   281.5  2170.7
     298 2164.34   309.9 2160.59   323.8 2154.39   335.7 2146.01   342.9 2142.45
   359.4  2139.9   377.12140.169   390.2 2138.53   394.9 2138.95   397.7 2140.37
   402.6 2142.09   428.3 2144.16   483.7 2142.55     507 2141.07   523.6 2141.52
   545.5 2143.93   572.6 2145.24   611.8 2151.01   633.2 2156.59     646 2160.84
   661.4 2167.74   690.4 2177.05   711.7 2185.59   723.3 2191.21   749.4 2208.74
#Mann= 7 ,-1 , 0
       0      .1       0      10    .035       0     290      .1       0
   377.1    .045       0   397.7      .1       0  410.21     .04       0
  550.21      .1       0
#XS Ineff= 2 , 0
                          430.87         2172.61
Permanent Ineff=
       F       F
Bank Sta=377.1,397.7
XS Rating Curve= 0 ,0
Exp/Cntr=0.3,0.1

Type RM Length L Ch R = 1 ,17040   ,181.5,185.2,190.4
XS GIS Cut Line= 3
     2179382.166      222949.024     2179495.184      222625.641
     2179675.906      222278.502
#Sta/Elev= 30
       0 2256.51    23.7 2248.35    48.4 2238.85   135.3 2211.92   161.7 2202.25
   239.5 2178.08   286.4 2166.03   305.6 2160.18   329.4 2148.94   350.3 2141.04
   355.72138.218   362.4 2134.91   364.9 2134.83   369.8 2135.59   378.42138.302
   399.4 2138.84   410.5 2140.35   423.3  2140.7   435.4  2140.3   447.4  2138.1
   458.5  2137.1   480.7 2138.17   525.1 2138.31   547.3  2139.4   606.5 2145.65
   647.2 2152.44   668.9 2160.16   715.2 2172.46   728.6 2177.11   733.9 2179.81
#Mann= 5 ,-1 , 0
       0      .1       0   355.7    .045       0   378.4      .1       0
  382.56     .04       0  552.56      .1       0
#XS Ineff= 2 , 0
                          431.32            2155
Permanent Ineff=
       F       F
Bank Sta=355.7,378.4
XS Rating Curve= 0 ,0
Exp/Cntr=0.3,0.1

Type RM Length L Ch R = 1 ,16855   ,232,231.8,231.9
XS GIS Cut Line= 3
     2179397.968      222967.241     2179654.074      222708.422
     2179904.201      222444.001
#Sta/Elev= 30
       0 2258.67    53.2 2241.75      81 2232.01    99.1 2226.81   123.4    2218
   150.6 2206.59   176.1  2197.9   221.3 2183.58     268 2170.05     320 2151.91
   350.1 2141.04     366 2136.23   369.12134.531   375.5 2131.63   380.3 2130.88
   385.1 2131.78   392.32134.818   398.9 2137.01   407.4 2137.77   425.5 2137.71
   440.6 2135.81   468.5  2137.6   499.6 2140.67   521.9 2143.65   566.5  2147.4
   609.4 2153.27   642.3 2155.32     662 2155.05   705.5 2155.96   728.1 2159.45
#Mann= 6 ,-1 , 0
       0      .1       0     320     .04       0   369.1    .045       0
   392.3     .04       0  444.11     .06       0  464.11      .1       0
#XS Ineff= 2 , 0
                          415.64         2171.96
Permanent Ineff=
       F       F
Bank Sta=369.1,392.3
XS Rating Curve= 0 ,0
Exp/Cntr=0.3,0.1

Type RM Length L Ch R = 1 ,16623   ,282.5,283.8,280.3
XS GIS Cut Line= 3
     2179579.379      223123.715     2179829.648      222858.746
     2180075.437      222589.957
#Sta/Elev= 30
       0 2275.64    42.5 2259.34    77.5 2247.11   130.7 2227.58   158.7 2215.62
   200.3 2200.14   268.3 2169.41   290.9 2158.24   320.9 2142.11   330.4 2135.43
   341.72129.427   348.3  2126.8   353.5 2126.43   358.2 2127.18   364.5 2129.09
   388.5 2130.05   417.3 2133.65   439.4 2134.58     451 2133.81   456.2 2134.44
   471.9  2138.7   514.6 2155.32   532.3 2163.03   574.1 2172.76     595  2178.9
   610.8 2181.54   637.5 2188.25   664.7 2192.36   677.5  2195.8   728.7 2202.26
#Mann= 6 ,-1 , 0
       0      .1       0   341.7    .045       0   364.5      .1       0
  394.48     .04       0  484.48     .06       0  534.48      .1       0
Bank Sta=341.7,364.5
XS Rating Curve= 0 ,0
Exp/Cntr=0.3,0.1

Type RM Length L Ch R = 1 ,16340   ,217.1,220.6,225.1
XS GIS Cut Line= 3
     2179813.981      223328.961     2180042.075      223038.579
     2180267.725      222754.176
#Sta/Elev= 30
       0 2264.01    36.4  2256.3   132.4 2231.67   166.8 2220.13   192.5 2209.48
   201.8 2203.71   220.5 2193.62   236.7  2186.6     245 2181.76   262.6 2173.27
   290.9 2161.05   343.4 2135.73     356  2129.1   362.72126.582   378.6 2122.75
   382.7 2122.37   391.1 2122.77     402 2126.47   416.2 2129.28   445.6 2131.28
   474.9 2143.94   492.8 2153.06   525.1 2164.33   591.9 2178.99   621.5 2188.31
   638.2 2194.71   657.3 2201.06   673.6 2204.44   692.3 2209.95   732.3 2219.88
#Mann= 4 ,-1 , 0
       0      .1       0   362.7    .045       0     402     .04       0
  499.25      .1       0
#XS Ineff= 2 , 0
          355.19 2134.55  427.49         2132.12
Permanent Ineff=
       F       F
Bank Sta=362.7,402
XS Rating Curve= 0 ,0
Exp/Cntr=0.3,0.1

Type RM Length L Ch R = 1 ,16119   ,202.9,201.9,200.9
XS GIS Cut Line= 3
     2179922.869      223422.583     2180200.742       223187.46
     2180478.614      222952.337
#Sta/Elev= 30
       0 2242.12    34.3 2233.24   100.8 2219.99     174 2198.86   302.8 2151.69
   311.4 2147.09   324.3 2142.75   346.7 2133.02   360.72122.629   364.8 2120.69
   371.8 2120.03   378.8  2120.4   383.72123.074   388.1 2125.46   393.1 2126.23
   420.7 2127.35     436 2123.78   462.6 2120.78     494 2128.06   506.8 2132.92
     522 2135.12   530.1 2138.94   558.1 2147.64   570.2 2153.29   583.7 2156.86
   607.9 2165.21   620.8 2168.01   642.3 2172.19   663.8 2174.49     728 2177.11
#Mann= 4 ,-1 , 0
       0      .1       0   360.7    .045       0   383.7     .04       0
     494      .1       0
#XS Ineff= 2 , 0
                          439.86         2135.23
Permanent Ineff=
       F       F
Bank Sta=360.7,383.7
XS Rating Curve= 0 ,0
Exp/Cntr=0.3,0.1

Type RM Length L Ch R = 1 ,15917   ,205.1,207.3,207
XS GIS Cut Line= 2
     2180049.003      223613.488     2180616.711      223068.349
#Sta/Elev= 30
       0 2217.89    95.6  2191.8   117.1 2184.84   154.2 2174.45   262.7 2146.16
   313.9 2134.66   358.4 2126.83   386.3    2124   393.52121.019   407.1 2118.04
   411.8 2118.89  415.52 2120.73   418.7 2122.46   423.4 2123.62   445.8 2124.58
   453.6  2124.4   473.1 2121.48     490 2121.21   504.2 2122.06     514 2120.89
   532.7 2120.67   546.4 2119.29   617.9 2122.68   643.8 2129.19   659.6 2131.89
   687.9 2135.12   705.1 2135.35   718.7 2136.79   750.5 2146.38   787.1 2154.29
#Mann= 7 ,-1 , 0
       0      .1       0     350    .035       0   393.5    .045       0
  415.52     .06       0     490      .1       0     550    .035       0
     620      .1       0
#XS Ineff= 2 , 0
                          434.36         2151.23
Permanent Ineff=
       F       F
Bank Sta=393.5,415.52
XS Rating Curve= 0 ,0
Exp/Cntr=0.3,0.1

Type RM Length L Ch R = 1 ,15710   ,178.7,178,176.8
XS GIS Cut Line= 3
     2180187.161      223727.587     2180466.168      223493.825
     2180747.125      223262.317
#Sta/Elev= 30
       0 2186.73    56.2  2168.6    68.1 2165.78   133.1 2145.97   215.7 2132.49
   244.8 2128.74   333.2 2121.54     359 2120.89   367.32118.787   371.9 2116.83
   376.2 2116.36   380.4 2116.67  385.342118.807   391.6  2121.3   410.3 2122.04
   424.2 2121.73   436.1 2119.04   452.7 2117.58   482.4  2118.7   503.5 2118.12
   554.7 2119.46   585.7 2119.36   610.7 2117.72   636.3 2118.23     648 2121.54
   669.5 2134.69   682.9  2144.6   699.2 2154.06   715.5 2162.18     728  2167.2
#Mann= 7 ,-1 , 0
       0      .1       0     150    .035       0     320     .04       0
   367.3    .045       0  385.34     .04       0  473.99     .06       0
  623.99      .1       0
#XS Ineff= 2 , 0
                          418.66         2156.63
Permanent Ineff=
       F       F
Bank Sta=367.3,385.34
XS Rating Curve= 0 ,0
Exp/Cntr=0.3,0.1

Type RM Length L Ch R = 1 ,15532   ,175.6,186.7,197.6
XS GIS Cut Line= 3
     2180206.198      223749.696     2180529.906      223677.724
     2180850.108      223376.901
#Sta/Elev= 30
       0 2180.88    17.1  2173.5    27.2 2170.49    77.6 2150.92   107.9 2141.93
   154.9 2131.81   203.7 2126.33   242.2  2123.6   289.4 2119.34   388.4 2116.67
   397.7 2117.55  404.912115.935   410.1 2114.09   413.9 2113.84   418.6 2114.43
   423.42116.265   439.5 2119.64   446.4 2120.12   468.6 2119.66   478.9 2118.09
   485.9 2116.06   489.9  2115.8   536.9  2116.8   599.2 2116.71   617.2 2120.79
   630.7 2129.66   671.2 2150.43   715.1 2166.48   724.9 2170.54     771 2183.91
#Mann= 5 ,-1 , 0
       0      .1       0     120    .035       0  404.91    .045       0
   423.4     .06       0  561.61      .1       0
#XS Ineff= 2 , 0
                          458.01         2154.59
Permanent Ineff=
       F       F
Bank Sta=404.91,423.4
XS Rating Curve= 0 ,0
Exp/Cntr=0.3,0.1

Type RM Length L Ch R = 1 ,15345   ,226.8,233,233.2
XS GIS Cut Line= 3
     2180228.522      223801.668     2180739.975      223755.849
      2181059.42      223780.155
#Sta/Elev= 30
       0 2169.09      24 2160.77    47.1 2151.81      57 2149.03    76.7 2142.38
   103.3 2136.84   132.7  2131.7     169  2127.3   244.2 2121.15     304 2118.33
   367.2 2114.08   452.2 2114.96   465.4 2114.68   474.2 2113.46     484 2111.24
   488.5 2110.82   491.8 2111.01   495.1 2112.12   497.22113.792   501.7 2116.97
   511.2 2118.02   547.7 2118.16   583.9 2116.82   636.6 2119.94   646.4 2122.92
   715.5 2139.08   794.5 2147.25     811 2150.67   827.1 2152.82   833.9 2154.26
#Mann= 6 ,-1 , 0
       0      .1       0     170    .035       0     470     .06       0
   474.2    .045       0   497.2     .06       0   663.5      .1       0
Bank Sta=474.2,497.2
XS Rating Curve= 0 ,0
Exp/Cntr=0.3,0.1

Type RM Length L Ch R = 1 ,15112   ,356,348.4,332.4
XS GIS Cut Line= 3
     2180231.295      223896.474     2180904.906      223932.932
     2181064.628      223837.446
#Sta/Elev= 30
       0 2160.99    40.9 2148.03      54 2142.29   103.3 2132.61   139.5 2128.78
   226.7 2122.31     284 2119.13     330 2113.64   337.12110.807   343.2 2108.47
     353 2109.02     3572110.788   362.9 2112.59   448.6 2110.64   494.3 2111.42
   612.6 2111.02   625.8 2109.33   645.5 2109.97     660 2114.67   671.7 2116.56
   698.4 2116.06   701.9 2116.85   705.7 2119.27   718.2 2130.64   732.4 2139.35
   744.1 2145.13   759.2  2148.9   784.5 2152.97     828 2158.07   860.7 2159.84
#Mann= 6 ,-1 , 0
       0    .035       0   337.1    .045       0     357    .035       0
     570     .06       0     660     .08       0   704.6      .1       0
#XS Ineff= 2 , 0
                          569.99          2147.5
Permanent Ineff=
       F       F
Bank Sta=337.1,357
XS Rating Curve= 0 ,0
Exp/Cntr=0.3,0.1

Type RM Length L Ch R = 1 ,14764   ,146.7,142.4,136.6
XS GIS Cut Line= 2
     2180385.809      224410.363     2181078.517       223866.96
#Sta/Elev= 30
       0 2128.93   104.4 2120.27   171.9 2118.97   237.6 2116.36   276.7 2109.24
   293.4 2109.08   327.32106.339   338.1 2103.44  348.762106.232   352.6 2107.63
   356.8 2107.93   368.4 2106.99   401.2 2106.36   496.2 2106.17   533.4 2107.43
   651.2 2108.32   672.8 2109.14   677.4 2109.82   689.5 2114.31   697.8 2115.83
     727 2115.97     730 2116.79     746 2127.29   752.1 2132.52   761.9 2143.07
   765.7 2145.81   772.9 2149.26   781.2 2151.81   814.8 2155.73   880.4 2159.67
#Mann= 7 ,-1 , 0
       0    .035       0   327.3    .045       0  348.76    .035       0
     520     .06       0     650     .08       0     770     .04       0
     800      .1       0
#XS Ineff= 2 , 0
          317.32 2108.35  498.88         2109.25
Permanent Ineff=
       F       F
Bank Sta=327.3,348.76
XS Rating Curve= 0 ,0
Exp/Cntr=0.5,0.3

Type RM Length L Ch R = 1 ,14621   ,49.7,49.5,50.5
XS GIS Cut Line= 3
     2180573.309      224550.988     2180948.309      224018.002
     2181088.934      223899.946
#Sta/Elev= 30
       0 2113.07      61 2110.57   156.4 2109.37   184.6    2107   201.1 2106.34
   277.6 2106.47   281.6 2106.07  286.14 2103.45   291.9 2100.74   297.6 2100.29
   301.7 2100.64   311.1 2103.63   345.8 2103.67   366.1 2104.62   480.1 2104.82
   510.3 2106.12   588.4 2106.34   615.5 2109.71   639.1 2110.67   664.1 2115.38
   676.5 2116.04   696.3 2115.89   701.4 2117.99   718.4 2129.39   725.4 2135.13
     732 2142.15   736.9 2146.63   741.2 2148.49   762.6 2152.11   835.3 2159.24
#Mann= 7 ,-1 , 0
       0    .035       0  286.14    .045       0   311.1    .035       0
     530     .06       0     650     .08       0  711.69     .04       0
  801.69      .1       0
#XS Ineff= 4 ,-1
  139.52  276.98 2110.32  276.98  285.422104.302   312.7  374.29 2104.32
  375.86   598.8 2110.56
Permanent Ineff=
       F       F       F       F
Bank Sta=286.14,311.1
XS Rating Curve= 0 ,0
Exp/Cntr=0.5,0.3

Type RM Length L Ch R = 1 ,14572   ,148.2,144.5,134.6
XS GIS Cut Line= 3
     2180623.656      224573.557     2180988.239      224031.891
     2181104.559      223932.932
#Sta/Elev= 30
       0 2109.63    82.6 2107.85   236.2  2106.7   265.3 2104.32   281.1 2104.31
   287.32102.261   292.9 2100.03   296.9 2099.34   308.8 2099.71   316.7 2102.23
   326.1 2103.44   352.3 2103.12   363.5 2101.98   373.3 2103.81     397 2104.42
   506.5 2104.77   567.2  2106.2   580.9 2107.52   597.9 2110.78   621.2 2113.18
   654.6 2115.68   678.2 2115.51   683.2 2117.43   707.8 2132.71   712.8  2136.6
   720.7 2144.38   726.7 2147.86   746.5 2151.64   780.3  2155.5   805.7 2157.34
#Mann= 6 ,-1 , 0
       0    .035       0   287.3    .045       0   316.7    .035       0
     480     .06       0  672.93     .04       0  782.93      .1       0
#XS Ineff= 3 ,-1
       0  282.23 2104.03  322.97     346 2103.74  346.58  409.44 2105.38
Permanent Ineff=
       F       F       F
Bank Sta=287.3,316.7
XS Rating Curve= 0 ,0
Exp/Cntr=0.5,0.3

Type RM Length L Ch R = 1 ,14427   ,181.3,183.7,186
XS GIS Cut Line= 3
       2180818.1      224707.238     2180963.934      224226.335
     2181142.753       223991.96
#Sta/Elev= 30
       0  2106.6    74.8 2103.08   174.7 2101.24   222.3 2101.31   242.8  2100.3
     308 2099.47     332 2099.52   349.1 2100.69   366.2 2100.32   379.8 2101.28
     385 2100.67   393.7 2097.47     401 2098.32     404  2099.1  406.552100.708
   410.8 2102.83   414.1 2103.18     428 2102.53   490.4 2102.58     552 2104.24
   584.4 2106.29     648  2114.6   676.7  2115.1   690.7 2124.18   714.1 2134.93
   718.8 2137.99   723.5 2141.96   726.4 2143.56   767.9 2150.34   797.3 2153.14
#Mann= 5 ,-1 , 0
       0    .035       0     385    .045       0  406.55    .035       0
  522.53     .06       0  712.53      .1       0
#XS Ineff= 2 , 0
          269.36 2131.34
Permanent Ineff=
       F       F
Bank Sta=385,406.55
XS Rating Curve= 0 ,0
Exp/Cntr=0.3,0.1

Type RM Length L Ch R = 1 ,14244   ,207.6,215.6,211
XS GIS Cut Line= 3
     2180934.854      224806.703     2181139.281      224288.835
     2181274.697      224158.627
#Sta/Elev= 30
       0 2102.68    28.2 2102.11    42.8 2100.92   162.8 2097.92   212.8 2097.89
   307.4 2099.93   406.1  2096.9   434.4 2096.87   468.32097.892   476.7 2095.61
   483.4 2095.43   488.5 2095.77   497.8 2097.65   508.4 2096.75   522.5  2096.6
   526.1 2097.99   529.6 2100.65   536.6 2107.42     539 2108.83   547.2 2110.53
   584.6 2113.13   605.4  2112.6   638.6 2112.77   643.4 2114.69   654.2 2124.35
   658.8 2126.91   679.7 2132.01   690.7 2133.52   728.3 2140.77   744.6 2143.09
#Mann= 5 ,-1 , 0
       0    .035       0     430      .1       0   468.3    .045       0
   497.8      .1       0     530     .04       0
#XS Ineff= 2 , 0
          304.67 2121.07
Permanent Ineff=
       F       F
Bank Sta=468.3,497.8
XS Rating Curve= 0 ,0
Exp/Cntr=0.3,0.1

Type RM Length L Ch R = 1 ,14028   ,220.8,236.4,243.9
XS GIS Cut Line= 3
     2181032.076       224896.98     2181264.281      224457.238
     2181479.559      224300.988
#Sta/Elev= 30
       0 2099.38      21 2098.69    38.9 2097.09    80.4 2096.07   213.4 2096.15
   291.8 2097.38   343.8 2096.74   380.9 2094.29     408 2094.37   432.8 2095.43
   438.42094.961   446.8 2091.55   452.3 2090.95     459 2091.38  469.412095.045
   499.7  2101.6   528.7 2105.55   551.8 2107.74   561.2 2107.76   568.6  2108.5
   596.5 2108.23   601.2 2110.33   608.2 2115.04   612.9 2117.36   629.4 2118.24
   638.7 2122.86   644.6 2124.31   661.9 2126.39   713.9 2136.11   763.3 2143.15
#Mann= 5 ,-1 , 0
       0    .035       0   438.4    .045       0  469.41    .035       0
  577.28     .04       0  647.28      .1       0
#XS Ineff= 2 , 0
          360.15 2125.05
Permanent Ineff=
       F       F
Bank Sta=438.4,469.41
XS Rating Curve= 0 ,0
Exp/Cntr=0.3,0.1

Type RM Length L Ch R = 1 ,13792   ,176.4,183.3,165.8
XS GIS Cut Line= 3
     2181104.993       224959.48      2181349.35       224679.46
     2181745.358      224433.276
#Sta/Elev= 30
       0 2097.67    57.8  2094.7   141.5 2093.58   222.9 2093.41   271.7 2094.73
   367.1 2094.37   378.1 2093.85   398.8 2091.39   423.6 2091.72     436 2089.93
   453.22089.612   471.8 2089.09   481.3 2087.99   486.1  2088.7     4892090.158
   493.2 2091.93   501.7 2092.97   514.6 2099.37     523 2101.43     579 2103.03
   598.3 2105.28   614.7 2107.99   625.3 2110.49   652.8 2110.74   657.6 2111.83
   671.7 2117.11   705.2 2121.88   777.8 2137.41   800.5 2139.86   837.9 2140.86
#Mann= 5 ,-1 , 0
       0    .035       0   453.2    .045       0     489    .035       0
  511.65     .04       0  641.65      .1       0
Bank Sta=453.2,489
XS Rating Curve= 0 ,0
Exp/Cntr=0.3,0.1

Type RM Length L Ch R = 1 ,13608   ,243,249.4,251.3
XS GIS Cut Line= 3
     2181302.475      225068.349     2181543.795      224714.182
     2181789.701       224478.42
#Sta/Elev= 30
       0 2092.96    31.3 2091.02    75.2  2090.4   138.5 2090.09     214 2091.28
   287.7 2088.55   327.8 2089.31   343.8 2087.64   349.1 2085.58   353.8 2084.87
     373 2087.94   380.7 2089.18   391.6 2089.05   416.4 2090.68     433  2090.9
   439.5 2091.95   450.2 2096.73   457.2 2098.63   471.3 2099.22     499 2098.92
   559.3 2104.63   570.5 2107.83   596.4  2109.5   607.6 2109.33   625.8 2117.39
   635.9 2118.91   674.8  2127.3   707.8 2130.39   748.5 2131.43   769.2 2133.26
#Mann= 5 ,-1 , 0
       0    .035       0   343.8    .045       0     373    .035       0
  438.57     .04       0  578.57      .1       0
#XS Ineff= 2 , 0
          300.76 2094.61  389.15         2092.13
Permanent Ineff=
       F       F
Bank Sta=343.8,373
XS Rating Curve= 0 ,0
Exp/Cntr=0.3,0.1

Type RM Length L Ch R = 1 ,13359   ,243.2,244.1,242.8
XS GIS Cut Line= 3
      2181392.01      225143.684      2181674.46      224909.576
     2181951.949       224674.78
#Sta/Elev= 30
       0 2090.56    19.9 2089.61    94.4 2088.06   287.2 2088.78   377.9 2086.42
   382.2 2085.83  384.482084.618   389.7  2080.9   395.1  2079.8   399.9 2080.03
     408 2081.54  411.55  2084.3   415.9 2088.07   420.9 2090.93   425.2 2092.38
   432.2 2092.97   446.7 2092.99   455.3 2092.33     471 2085.77   491.3 2083.65
   496.4 2083.95   506.5 2086.24     530 2088.12   541.2 2090.37   569.6 2098.75
   618.4 2108.68   639.4    2110   660.3 2115.39   689.4 2118.68   730.4 2124.96
#Mann= 5 ,-1 , 0
       0    .035       0  376.86     .04       0  384.48    .045       0
  411.55     .04       0  506.86      .1       0
#XS Ineff= 2 , 0
          308.45 2092.69  442.88         2101.22
Permanent Ineff=
       F       F
Bank Sta=384.48,411.55
XS Rating Curve= 0 ,0
Exp/Cntr=0.3,0.1

Type RM Length L Ch R = 1 ,13115   ,237.7,237.6,236.7
XS GIS Cut Line= 3
     2181567.044      225318.513     2181844.136      225082.471
     2182121.229      224846.429
#Sta/Elev= 30
       0 2086.73    56.9 2089.15   127.2 2083.79   213.2 2080.72   258.8    2080
   354.8 2082.22   366.5 2081.96   370.6 2080.93   380.6 2076.74   387.4 2077.83
   393.5 2081.45     399    2084     406 2085.85   423.7 2087.08   438.6 2086.51
   449.6 2085.08   458.2 2082.82   486.4 2082.46   516.8 2080.15   550.3  2082.4
   564.3 2081.99   580.6 2080.08   591.8 2085.31   606.2 2090.35   620.1 2099.44
   624.8 2101.45   643.5 2106.54   666.7 2106.94   696.9  2112.1     728 2121.77
#Mann= 5 ,-1 , 0
       0    .035       0     340     .04       0   370.6    .045       0
   393.5     .04       0     494      .1       0
#XS Ineff= 2 , 0
          252.21 2105.97  420.68         2113.32
Permanent Ineff=
       F       F
Bank Sta=370.6,393.5
XS Rating Curve= 0 ,0
Exp/Cntr=0.3,0.1

Type RM Length L Ch R = 1 ,12877   ,248.8,261.2,269.7
XS GIS Cut Line= 2
     2181725.563      225506.678     2182273.127      225016.819
#Sta/Elev= 30
       0 2081.89    26.4 2082.07    56.9 2081.22   174.7  2082.7   224.5 2082.75
   281.7 2081.86   307.8 2080.49   340.4 2077.35   352.2 2077.12   365.4 2077.78
   367.32077.421   375.2 2074.38   377.6 2074.06   391.8 2075.77   400.22077.402
   409.4 2080.04   419.4 2081.08   440.4 2080.83   460.1 2077.07   568.3 2079.04
   612.2 2082.23   629.5  2084.7   642.4 2087.34     661 2092.73   686.4 2102.76
   691.2 2103.67   705.2 2103.89     711  2105.9   726.3 2112.81   734.7 2114.42
#Mann= 6 ,-1 , 0
       0    .035       0     340     .04       0   367.3    .045       0
   400.2     .04       0     460     .06       0     610      .1       0
#XS Ineff= 2 , 0
                          423.71         2103.48
Permanent Ineff=
       F       F
Bank Sta=367.3,400.2
XS Rating Curve= 0 ,0
Exp/Cntr=0.3,0.1

Type RM Length L Ch R = 1 ,12616   ,73.8,84.4,97.4
XS GIS Cut Line= 2
     2181745.184      225544.043     2182469.142      225391.266
#Sta/Elev= 30
       0 2081.06    50.3 2080.65    83.9  2079.9   153.5 2079.75   194.5 2079.02
   221.4 2079.43   281.7 2078.49   342.1 2079.05   362.2 2077.68   382.3 2075.28
   392.4 2073.47   405.8 2073.97   412.52073.491     436 2071.11     442  2073.3
     446 2074.28   466.1 2074.73   482.9 2077.45   495.3 2078.48   517.5 2078.38
   523.3 2077.58   533.2 2074.88   536.5 2074.38   545.2 2074.98   633.8 2076.26
   677.4 2078.41   694.1 2080.77   707.6 2083.69   724.3 2089.46   739.9 2098.17
#Mann= 4 ,-1 , 0
       0    .035       0   412.5    .045       0     442     .06       0
   739.9    .035       0
#XS Ineff= 2 , 0
                           503.4         2091.51
Permanent Ineff=
       F       F
Bank Sta=412.5,442
XS Rating Curve= 0 ,0
Exp/Cntr=0.3,0.1

Type RM Length L Ch R = 1 ,12532   ,51.4,51.7,51.5
XS GIS Cut Line= 3
     2181759.072      225563.141      2182099.35      225505.849
      2182434.42      225649.946
#Sta/Elev= 30
       0  2080.7    53.5 2080.35    92.3 2079.21    99.1 2079.15   109.6 2079.49
   165.6 2079.06   205.6 2078.17   218.9 2078.22   265.4 2077.29   318.7 2077.42
   325.3 2077.92   345.1  2076.9   365.8 2075.04   377.4 2074.29   391.7 2072.48
   416.7 2072.13   424.5 2071.45     431 2071.21     446 2072.08     457 2072.63
     467 2072.57   478.6 2072.98   513.2 2073.07   553.8 2073.74   577.4 2075.65
   596.9 2075.93   617.1    2077     656 2079.86   677.4 2080.54   709.8 2080.73
#Mann= 6 ,-1 , 0
       0    .035       0   416.7    .045       0     446     .04       0
  535.07     .06       0  575.07    .035       0  645.07     .04       0
#XS Ineff= 3 ,-1
       0   416.7  2072.8     446     540  2072.8  542.13   633.4 2075.98
Permanent Ineff=
       F       F       F
Bank Sta=416.7,446
XS Rating Curve= 0 ,0
Exp/Cntr=0.3,0.1
